--- WhtdyCrk.prj (project) ---

Proj Title=WhtdyCrk
Current Plan=p01
Default Exp/Contr=0,0
English Units
Geom File=g01
Flow File=f01
Plan File=p01
BEGIN DESCRIPTION:
END DESCRIPTION:
DSS Export Rating Curves= 0
DSS Export Rating Curve Sorted= 0
DSS Export Volume Flow Curves= 0
DXF OffsetX= 0
DXF OffsetY= 0
DXF ScaleX= 0
DXF ScaleY= 0

--- WhtdyCrk.p01 (plan) ---

Plan Title=Floodplain
Program Version=4.00
Geom File=g01
Flow File=f01
K Sum by GR=0
Std Step Tol=0.01
Critical Tol=0.01
Num of Std Step Trials=20
Max Error Tol=0.3
Flow Tol Ratio=0.001
Split Flow NTrial=30
Split Flow Tol=0.02
Split Flow Ratio=0.02
Log Output Level=0
Friction Slope Method=1
Unsteady Friction Slope Method=2
Unsteady Bridges Friction Slope Method=1
Global Log Level=0
CheckData=False
Run HTab=0
Run UNet=0
Run PostProcess=0
UNET Theta=0
UNET Theta Warmup=0
UNET ZTol=0
UNET ZSATol=0
UNET MxIter=0
UNET MaxInSteps=0
UNET DtIC=0
UNET DtMin=0
UNET MaxCRTS=0
UNET WFStab=0
UNET SFStab=0
UNET WFX=0
UNET SFX=0
UNET DSS MLevel=0
UNET DZMax Abort=0
UNET Convert EG Bridges=0
UNET Use Existing IB Tables=0
UNET Froude Limit=0
UNET Froude Power=0
Write IC File=0
Echo Input=False
Echo Output=False
Write Detailed=0

--- WhtdyCrk.f01 (steady flow) ---

Flow Title=NFF Regression Equation
Program Version=4.00
Number of Profiles=1
Profile Names=P100yr
River Rch & RM=WhtdyCrk,Main      ,58033.9
1356.159
River Rch & RM=WhtdyCrk,Main      ,57631.2
2234.733
River Rch & RM=WhtdyCrk,Main      ,52433.9
2397.153
River Rch & RM=WhtdyCrk,Main      ,43233.9
2639.999
River Rch & RM=WhtdyCrk,Main      ,42761.3
2957.697
River Rch & RM=WhtdyCrk,Main      ,41594.8
3104.094
River Rch & RM=WhtdyCrk,Main      ,33315.8
3441.475
River Rch & RM=WhtdyCrk,Main      ,32833.9
3878.502
River Rch & RM=WhtdyCrk,Main      ,29233.9
4118.129
River Rch & RM=WhtdyCrk,Main      ,23626.6
4520.971
River Rch & RM=WhtdyCrk,Main      ,16875.5
4807.349
River Rch & RM=WhtdyCrk,Main      ,89
5236.833
River Rch & RM=WhtdyCrk,Main      ,89
5237.940
Boundary for River Rch & Prof#=WhtdyCrk,Main      ,1
Up Type=0
Dn Type=3
Dn Slope=0.004246

--- WhtdyCrk.g01 (geometry) ---

Geom Title=USGS 3m DEM
Program Version=4.00

River Reach=WhtdyCrk        ,Main
Reach XY= 30
     1833899.572      340217.437       1833615.2      342747.989
     1834363.926      343827.883     1833892.372      344558.611
     1834439.519       346002.07     1835289.035      346973.975
     1836397.727      346865.985     1837412.827      347492.324
       1836377.6      351424.376     1835523.548      352434.025
     1834047.109      352959.596     1834140.467       354066.06
     1833493.877       355179.44     1829995.918      356973.563
     1830191.773      358166.894     1828355.587      360007.467
     1826103.164      359367.877     1825658.046      360135.422
      1824042.37      360172.709     1823992.917      361723.009
     1822400.142      362703.549     1823121.183      365329.351
      1819633.77      366423.101     1819460.158      366828.917
      1817604.69      366657.476     1815792.624      368031.174
     1814158.509      369917.025     1814698.874       370782.91
     1816658.509      370698.275     1815291.322       372970.41

Type RM Length L Ch R = 1 ,58033.9 ,167.574,156.025,150.22
XS GIS Cut Line= 3
      1833429.25      340273.353     1833903.196      340226.757
     1834323.766      340063.202
#Sta/Elev= 30
       0 1553.55    19.4 1544.11    29.2 1542.16    48.6 1533.08    58.3 1530.93
    77.8 1522.11    87.5 1519.57   106.9 1511.43   116.6 1509.14   136.1 1501.09
   165.2 1491.25   184.7 1486.25     243 1480.19   330.4  1466.2   466.5 1460.66
   468.7 1460.82   483.7  1462.1   505.7  1467.1   584.1 1465.97     643 1478.14
   672.4 1482.66   731.3 1486.76   750.9 1489.07   770.5 1493.28     800 1496.67
   819.6  1496.5   839.2 1494.68   868.6 1489.26   888.2 1487.19   927.5 1487.24
#Mann= 3 , 0 , 0
       0      .1       0   468.7    .045       0   483.7      .1       0
Bank Sta=468.7,483.7
XS Rating Curve= 0 ,0
Exp/Cntr=0.3,0.1

Type RM Length L Ch R = 1 ,57877.9 ,227.994,246.716,262.247
XS GIS Cut Line= 4
     1833399.024      340499.791     1833889.699      340381.213
     1834082.029      340325.307     1834314.548      340121.075
#Sta/Elev= 30
       0 1589.53    48.5    1575   155.3    1548   174.7 1541.17   203.9 1533.04
   213.6  1531.4   242.7 1522.14   281.5 1512.36   300.9 1505.37   349.5 1492.22
   368.9 1485.61   378.6 1483.53     398 1476.42   407.7 1474.69   427.1 1467.75
   456.3 1463.11     543 1460.77     558 1460.54     562 1460.53   619.3 1464.07
     686  1462.6   714.8 1466.08   850.2 1467.36   869.5 1470.09   888.8 1474.84
   898.5 1475.33   927.5 1481.78   985.6 1487.38  1004.9 1486.99  1014.6 1485.72
#Mann= 3 , 0 , 0
       0      .1       0     543    .045       0     558      .1       0
Bank Sta=543,558
XS Rating Curve= 0 ,0
Exp/Cntr=0.3,0.1

Type RM Length L Ch R = 1 ,57631.2 ,484.554,489.736,497.41
XS GIS Cut Line= 3
     1833432.408      340536.989     1833936.262      340567.871
     1834542.629      340577.238
#Sta/Elev= 30
       0 1583.22    19.4 1577.84    58.2 1570.12    77.7 1564.64   106.8 1558.13
   116.5 1557.07   135.9 1550.76   174.7 1541.19   203.9 1531.71   213.6 1530.38
   262.1 1515.65   291.2 1508.07   330.1 1502.87   339.8 1500.56   368.9 1491.99
   407.7 1476.54   436.8 1466.86   446.6 1464.74   490.9 1461.74   504.8 1460.61
   505.9 1460.63   592.8 1468.06   671.1 1472.82   739.6 1487.11   778.7 1491.99
   827.6 1492.43   925.4 1488.08   974.3  1490.1    1033 1497.15  1111.2 1510.49
#Mann= 3 , 0 , 0
       0      .1       0   490.9    .045       0   505.9      .1       0
Bank Sta=490.9,505.9
XS Rating Curve= 0 ,0
Exp/Cntr=0.3,0.1

Type RM Length L Ch R = 1 ,57141.5 ,305.648,307.524,302.47
XS GIS Cut Line= 3
      1833454.69      340897.963     1833888.006      341027.229
     1834354.797      341160.859
#Sta/Elev= 30
       0 1557.88    39.3  1553.5    98.3 1540.49   127.8 1532.34   186.8 1519.39
   235.9 1510.11   265.4 1502.27   344.1 1477.57   353.9 1476.01   373.5 1468.21
   383.4 1465.87   393.2 1465.42   452.2 1468.58   461.9 1468.31   470.8 1466.11
   485.8 1460.21   500.7 1456.32   520.2 1458.25   549.3 1464.18   568.7 1471.03
   578.4 1472.72   597.8  1479.2   607.6 1480.78   675.5 1500.83     695 1508.48
   753.2 1527.36   762.9 1528.69   792.1 1539.59     860 1547.46   937.7 1552.29
#Mann= 3 , 0 , 0
       0      .1       0   470.8    .045       0   485.8      .1       0
#XS Ineff= 2 , 0
           453.5 1468.26
Permanent Ineff=
       F       F
Bank Sta=470.8,485.8
XS Rating Curve= 0 ,0
Exp/Cntr=0.3,0.1

Type RM Length L Ch R = 1 ,56833.9 ,418.674,400,389.817
XS GIS Cut Line= 3
     1833408.754      341085.215     1833808.758      341304.465
     1834276.992      341429.914
#Sta/Elev= 30
       0 1538.32   126.2  1512.2   194.1 1502.02   242.6 1495.76     262 1492.29
   271.7 1491.57   291.2 1487.37   310.6 1484.66   349.4  1476.2   359.1  1472.9
   368.8 1471.34   397.9 1463.34   417.3 1460.39     427    1458   446.4 1455.74
   448.7 1455.76   463.7 1456.32   504.6 1459.72   533.7 1465.05   553.1  1465.9
   582.2 1462.68   601.6 1466.86     621 1472.82   630.7 1474.62   717.9  1499.1
   766.4 1508.99   785.8 1515.37   795.5 1517.14     873 1543.43   940.9 1554.35
#Mann= 3 , 0 , 0
       0      .1       0   448.7    .045       0   463.7      .1       0
#XS Ineff= 2 , 0
                          551.82         1465.58
Permanent Ineff=
       F       F
Bank Sta=448.7,463.7
XS Rating Curve= 0 ,0
Exp/Cntr=0.3,0.1

Type RM Length L Ch R = 1 ,56433.9 ,387.002,400,402.954
XS GIS Cut Line= 3
     1833356.746      341811.523     1833801.022       341662.76
     1834273.547      341535.479
#Sta/Elev= 30
       0 1583.14    87.8 1570.74   107.4 1564.52   117.1  1563.3   146.4 1553.94
   165.9 1544.86   185.5 1538.21   195.2 1533.12   263.5 1507.62   273.3 1506.37
   292.8  1500.1   341.6 1490.48   380.7 1475.67   390.4  1470.5   429.5 1461.51
     461 1456.06     476 1454.99   478.3 1454.92   497.9 1455.22   527.2 1459.07
   566.4 1460.04   576.2  1461.6   595.8 1468.04   615.3 1478.11   644.7 1486.92
   654.5 1487.99   674.1 1494.19   781.7 1516.98   899.2 1551.75   957.9 1561.23
#Mann= 3 , 0 , 0
       0      .1       0     461    .045       0     476      .1       0
Bank Sta=461,476
XS Rating Curve= 0 ,0
Exp/Cntr=0.3,0.1

Type RM Length L Ch R = 1 ,56033.9 ,394.567,400,409.855
XS GIS Cut Line= 3
     1833369.038      341919.818     1833900.479      342030.561
     1834339.862      341969.733
#Sta/Elev= 30
       0 1571.71    67.9 1561.86   106.6 1553.77   164.8 1535.35   184.2 1527.52
   193.9 1525.71   242.3 1507.06     252 1505.41   271.4 1496.04   319.9  1477.6
   339.3 1467.95     349 1465.43   368.4 1463.33   535.4 1455.27   550.4 1454.93
   562.1 1454.89   571.8 1455.42   629.6 1469.54   668.2 1480.73   716.4 1497.12
     755 1508.35   774.3 1515.88   783.9  1517.4   803.2 1525.17   812.9 1526.44
   841.8 1535.81   861.1 1544.08   870.7 1545.74   918.9 1562.69   986.4  1579.5
#Mann= 3 , 0 , 0
       0      .1       0   535.4    .045       0   550.4      .1       0
Bank Sta=535.4,550.4
XS Rating Curve= 0 ,0
Exp/Cntr=0.3,0.1

Type RM Length L Ch R = 1 ,55633.9 ,274.274,264.05,257.775
XS GIS Cut Line= 3
     1833279.598      342124.147     1833679.141      342283.964
     1834257.658       342422.38
#Sta/Elev= 30
       0 1550.34    39.1  1544.6      88 1532.27   107.6 1529.62   185.8 1512.95
   215.2 1508.13   234.7 1506.58   244.5 1504.76   283.6 1493.52   303.2 1488.87
   352.1  1473.5   361.9 1471.43     401  1457.2   410.8 1455.54   420.5 1455.19
   422.8 1455.32   437.8 1456.01   557.1 1457.94   596.1 1459.67   713.1 1483.06
   752.1 1488.41   771.6 1493.98   781.4 1495.28   800.9 1501.46   830.1 1507.31
   947.2 1525.36   976.4 1528.68   995.9 1532.17  1015.4  1538.8  1025.2 1540.55
#Mann= 3 , 0 , 0
       0      .1       0   422.8    .045       0   437.8      .1       0
Bank Sta=422.8,437.8
XS Rating Curve= 0 ,0
Exp/Cntr=0.3,0.1

Type RM Length L Ch R = 1 ,55369.9 ,695.139,690.461,681.858
XS GIS Cut Line= 3
     1833229.829      342554.952     1833677.261      342532.703
     1834251.668      342523.413
#Sta/Elev= 30
       0 1512.55    48.7  1506.2    87.6 1502.31   165.6 1489.15     185  1486.8
   214.3  1481.2     224 1478.21   243.5 1473.82   292.2 1460.87   321.4 1458.74
   444.3 1454.92   457.7 1454.71   459.3 1454.74   486.9 1456.01   506.4 1458.49
   545.4  1462.1   564.8 1465.29   574.6 1465.89   613.5 1472.75   623.3 1475.31
     633 1476.35   662.2 1483.43   720.6 1492.86   769.3 1495.63     818 1499.89
   866.7 1506.66   944.6 1515.75   973.8    1520    1003 1525.64  1022.5 1531.07
#Mann= 3 , 0 , 0
       0      .1       0   444.3    .045       0   459.3      .1       0
Bank Sta=444.3,459.3
XS Rating Curve= 0 ,0
Exp/Cntr=0.3,0.1

Type RM Length L Ch R = 1 ,54679.4 ,244,245.488,247.344
XS GIS Cut Line= 3
     1833566.574      343092.845     1834019.383      342938.555
     1834482.255      342777.556
#Sta/Elev= 30
       0 1522.76    48.8  1512.3    68.3  1509.5   146.4 1499.81   224.5 1491.78
   253.8    1487   341.7  1461.2     410 1449.18   424.4 1447.71   429.6 1447.25
   439.4 1447.57   478.4 1450.51   488.2 1452.83     498 1456.66   507.8 1458.93
   556.8 1476.67   586.2 1484.11   615.6  1487.6   654.8 1496.07     694 1503.11
   752.8 1507.12   772.4 1509.81   782.2 1513.27   821.4 1523.45   831.2 1524.68
   880.2 1535.54   899.8 1537.63   919.4 1542.69   929.2 1543.67   968.4 1551.59
#Mann= 3 , 0 , 0
       0      .1       0   424.4    .045       0   439.4      .1       0
Bank Sta=424.4,439.4
XS Rating Curve= 0 ,0
Exp/Cntr=0.3,0.1

Type RM Length L Ch R = 1 ,54433.9 ,298.342,301.086,303.206
XS GIS Cut Line= 3
     1833667.198      343290.739     1834110.001       343147.24
     1834566.108      343012.346
#Sta/Elev= 30
       0 1553.37    58.2 1545.05    87.3 1535.42   116.4 1521.17   135.8 1513.73
   271.5 1486.75   310.3 1474.45   329.7 1466.19   339.4 1464.91   358.8 1457.66
   378.2 1454.53     458 1451.02     473 1449.61   494.6 1446.16   533.4 1449.87
   562.5 1457.13     582 1465.98   649.9 1490.26   659.6 1491.85   688.7 1501.96
   708.1 1510.41   717.9 1512.51   785.8  1534.6   805.2 1543.18   814.9 1545.54
   834.3 1555.69   863.5 1565.64   873.2 1567.11   902.3 1576.38   941.1 1583.78
#Mann= 3 , 0 , 0
       0      .1       0     458    .045       0     473      .1       0
Bank Sta=458,473
XS Rating Curve= 0 ,0
Exp/Cntr=0.3,0.1

Type RM Length L Ch R = 1 ,54132.9 ,307.016,311.234,315.452
XS GIS Cut Line= 3
     1833708.983      343412.855      1834167.87      343435.954
      1834631.82      343345.522
#Sta/Elev= 30
       0 1566.48    48.9 1559.48    97.8 1549.06   166.2 1524.75   185.7 1515.93
   244.4 1501.98   283.5 1494.22   332.4  1476.5   342.2 1474.39     391 1455.16
   430.1 1448.88   481.9 1447.76   496.9 1447.82   546.3  1442.1   555.9 1442.23
   565.6 1444.72   604.2 1460.03   652.4 1475.45   671.7 1483.67   681.3 1485.74
   700.6 1494.67   719.9 1500.84   729.6 1505.36   739.2 1507.11   768.2 1519.48
   806.7 1532.33     826 1541.15   874.3 1559.17   883.9 1563.78   932.1 1580.22
#Mann= 3 , 0 , 0
       0      .1       0   481.9    .045       0   496.9      .1       0
Bank Sta=481.9,496.9
XS Rating Curve= 0 ,0
Exp/Cntr=0.3,0.1

Type RM Length L Ch R = 1 ,53821.6 ,474.47,482.79,484.008
XS GIS Cut Line= 3
     1833801.596      343746.551     1834340.871      343705.707
     1834777.714      343654.315
#Sta/Elev= 30
       0 1565.16    39.3 1555.99      59 1549.09    68.8 1547.26     118 1529.63
   127.8  1527.5   147.5  1519.4   196.7  1502.9   216.3 1494.32   255.7 1481.33
   275.3 1472.72   285.2 1470.34   334.3 1452.79   432.7 1447.53   452.9 1444.41
   467.9 1442.49   481.8 1441.43   501.5 1442.82   589.7 1459.86   667.9 1486.68
   746.1 1505.14   804.7 1522.13   824.3 1529.29   834.1 1531.14   853.6  1538.2
   882.9 1546.42   892.7 1547.91   912.3 1554.35   951.4 1563.26   980.7 1572.27
#Mann= 3 , 0 , 0
       0      .1       0   452.9    .045       0   467.9      .1       0
Bank Sta=452.9,467.9
XS Rating Curve= 0 ,0
Exp/Cntr=0.3,0.1

Type RM Length L Ch R = 1 ,53338.8 ,365.776,373.053,380.165
XS GIS Cut Line= 3
     1833805.215      343903.473     1834259.291      344128.654
     1834705.213      344146.403
#Sta/Elev= 30
       0 1539.14     9.7 1536.63    29.2 1527.97      78 1514.33    97.5 1506.36
   126.7 1497.19   146.2 1492.49   165.7 1484.94   253.4    1460   302.2 1444.61
   321.7 1442.15   341.1 1441.46   448.4  1441.4   505.3 1442.99   520.3 1441.41
   526.2 1440.76   574.8 1450.44   662.1 1480.02   671.8 1481.37   700.9 1489.25
   720.3 1496.55     730 1497.81   749.4 1504.21   788.2 1512.77   807.6 1519.46
   836.7 1525.38   875.5  1530.2   914.3 1538.17   933.7 1543.27   953.1 1550.49
#Mann= 3 , 0 , 0
       0      .1       0   505.3    .045       0   520.3      .1       0
Bank Sta=505.3,520.3
XS Rating Curve= 0 ,0
Exp/Cntr=0.3,0.1

Type RM Length L Ch R = 1 ,52965.8 ,556.446,531.837,516.614
XS GIS Cut Line= 3
     1833741.231      344137.711     1834079.975      344411.313
     1834595.362      344644.917
#Sta/Elev= 30
       0 1490.59    58.1 1474.34    87.1  1463.6   106.4 1459.55   154.8 1442.52
   164.5 1441.22   280.6 1437.18   396.7 1438.55   416.1  1436.8   425.7 1434.17
   435.4 1433.66   440.7  1434.1   484.2 1441.55   513.5 1449.49     533 1456.08
   542.8 1457.76   562.3 1465.71   581.8 1471.04   630.6 1489.63   640.3 1491.46
   659.8 1498.49   669.6 1500.69   718.4 1510.09   776.9 1514.75   796.4  1518.1
   815.9 1519.92   864.7 1530.25   952.5 1541.76   962.3 1545.07  1001.3 1554.42
#Mann= 3 , 0 , 0
       0      .1       0   425.7    .045       0   440.7      .1       0
Bank Sta=425.7,440.7
XS Rating Curve= 0 ,0
Exp/Cntr=0.3,0.1

Type RM Length L Ch R = 1 ,52433.9 ,397.008,400,400.359
XS GIS Cut Line= 3
      1833522.97      345011.414     1833935.518      344839.308
     1834388.339      344696.125
#Sta/Elev= 30
       0 1552.42    19.4 1546.48    58.3 1536.71    77.7 1530.52    87.5 1528.62
   126.3 1516.22   145.8 1508.64   155.5 1506.86   174.9 1499.93   184.6 1498.47
   204.1 1492.68   242.9 1484.29   291.5 1475.76   320.7 1468.61   340.1 1462.62
   388.7 1450.93   408.1 1444.01   417.9 1441.98   439.5 1435.19   454.5 1431.96
   476.1 1429.83   640.9 1435.14   679.6 1437.48   737.8 1442.81   795.9 1455.12
     825 1463.05   834.7 1464.41   863.8 1472.58   883.2 1479.89   921.9 1492.38
#Mann= 3 , 0 , 0
       0      .1       0   439.5    .045       0   454.5      .1       0
Bank Sta=439.5,454.5
XS Rating Curve= 0 ,0
Exp/Cntr=0.3,0.1

Type RM Length L Ch R = 1 ,52033.9 ,407.521,400,394.628
XS GIS Cut Line= 3
     1833678.188      345307.689     1834117.794      345180.616
     1834553.805      345043.831
#Sta/Elev= 30
       0 1553.74     9.7  1550.7    19.5 1549.44    58.4  1540.8    77.9 1534.63
   107.1 1520.62   136.3 1510.32   155.8 1505.47     185 1501.83   214.2 1495.58
   233.7 1488.84   243.4  1487.5   262.9 1480.25   272.6 1478.82   292.1 1472.54
   311.6 1467.74   321.3 1463.75   340.8  1458.1     370 1446.34   389.5 1435.87
   408.9 1431.36   450.1 1424.71   457.6 1424.63   465.1 1425.17   720.1 1442.24
   749.3 1446.82   797.9 1459.88   807.6 1461.09   875.7 1475.19   914.6 1485.88
#Mann= 3 , 0 , 0
       0      .1       0   450.1    .045       0   465.1      .1       0
Bank Sta=450.1,465.1
XS Rating Curve= 0 ,0
Exp/Cntr=0.3,0.1

Type RM Length L Ch R = 1 ,51633.9 ,386.715,400,411.68
XS GIS Cut Line= 3
     1833925.069      345779.806     1834321.935      345492.475
     1834750.586      345219.371
#Sta/Elev= 30
       0 1521.66     9.8 1518.11    19.6  1516.8    78.4 1500.46   107.8 1494.69
     147 1484.69   205.8    1467   254.8 1456.69   274.4 1450.73   284.2 1449.35
   313.6 1441.95   352.8 1435.09   482.5 1422.28   497.5 1421.01   509.5 1420.79
   587.7 1428.52   597.5 1430.64   636.6 1443.69   695.2 1453.98   753.9 1467.78
   773.4 1471.32   802.7 1474.51   832.1 1481.98   851.6 1490.31   871.2 1495.29
   890.7 1503.34   900.5 1505.15     920 1511.71   968.9 1520.61   998.2 1528.12
#Mann= 3 , 0 , 0
       0      .1       0   482.5    .045       0   497.5      .1       0
Bank Sta=482.5,497.5
XS Rating Curve= 0 ,0
Exp/Cntr=0.3,0.1

Type RM Length L Ch R = 1 ,51233.9 ,410.354,400,386.856
XS GIS Cut Line= 3
     1833960.181      345882.296     1834422.984      345844.426
     1834890.147      345812.003
#Sta/Elev= 30
       0  1526.3    48.4 1515.94    67.7 1507.84    77.4 1505.97   106.4 1497.54
   125.8 1490.86   174.1 1478.18   183.8 1474.67   203.2 1469.92   212.8 1466.58
   232.2 1462.16   309.6 1441.71   319.2 1440.25   338.6  1434.9   367.6 1428.78
   396.6 1424.18   456.9 1417.86   464.3 1417.44   471.9 1417.77   513.1 1424.47
   591.2 1428.86   620.4 1432.94   708.2 1448.29   747.3  1453.2   776.5  1459.1
   805.8 1466.57   825.3 1473.18   874.1 1485.49   883.9  1488.7   932.6 1499.96
#Mann= 3 , 0 , 0
       0      .1       0   456.9    .045       0   471.9      .1       0
Bank Sta=456.9,471.9
XS Rating Curve= 0 ,0
Exp/Cntr=0.3,0.1

Type RM Length L Ch R = 1 ,50833.9 ,399.492,400,399.831
XS GIS Cut Line= 3
     1834178.815      346439.022     1834565.525        346202.7
     1834933.742      345918.428
#Sta/Elev= 30
       0 1540.73     9.6 1538.83    48.2 1526.28    67.5 1517.75    96.4 1508.46
   115.7 1503.71   144.6 1493.23   183.2 1482.65   212.1 1471.23   260.4 1456.33
   289.3 1445.55   298.9 1443.44   318.2 1436.58   347.1 1428.58     405 1424.57
   445.7 1417.09   460.7 1415.23   462.9 1415.14   472.6 1415.59     492 1421.68
   501.7  1422.9   598.6 1427.35   676.1 1441.67   734.3 1454.02   753.6  1456.7
   792.4  1459.7   821.5 1466.63   840.9 1473.78   860.2 1477.79   918.4 1495.69
#Mann= 3 , 0 , 0
       0      .1       0   445.7    .045       0   460.7      .1       0
Bank Sta=445.7,460.7
XS Rating Curve= 0 ,0
Exp/Cntr=0.3,0.1

Type RM Length L Ch R = 1 ,50433.9 ,412.036,400,391.439
XS GIS Cut Line= 3
      1834446.55      346713.204     1834852.352      346478.593
     1835209.124      346200.136
#Sta/Elev= 30
       0  1493.9     9.8 1490.76    19.5 1489.29    39.1 1482.58    78.1 1471.79
    87.9 1470.42   185.5 1442.76   214.8 1437.48   371.1 1420.37   400.4 1414.42
   429.7 1415.94   461.2 1414.96   476.2 1413.79   488.4 1411.73   508.1 1410.87
   517.9 1411.13   527.8 1415.97   537.6 1423.94   547.4 1427.57   586.8  1435.9
   616.3 1443.59     636 1445.47   714.7 1460.37   744.2  1470.8   763.9 1475.25
   803.3 1489.19   822.9    1494   872.1 1511.15   901.6 1518.36   921.3 1525.83
#Mann= 3 , 0 , 0
       0      .1       0   461.2    .045       0   476.2      .1       0
Bank Sta=461.2,476.2
XS Rating Curve= 0 ,0
Exp/Cntr=0.3,0.1

Type RM Length L Ch R = 1 ,50033.9 ,411.069,400,387.732
XS GIS Cut Line= 3
     1834824.067      347168.258     1835061.168       346781.87
     1835330.853       346359.78
#Sta/Elev= 30
       0 1514.09    86.8 1487.21    96.5 1486.51   115.7 1481.16   144.7 1475.18
   173.6 1465.95   192.9 1463.15   212.2 1456.75   241.1 1450.42   270.1 1441.92
   279.7 1440.95   327.9 1430.69   385.8 1411.94     434 1408.96   445.8 1410.12
   460.8 1413.46   482.8 1415.31   551.5 1415.18     581 1417.68   620.3 1426.04
   649.8 1429.82   728.3 1443.95   806.9 1453.73   846.2  1461.7   865.8 1467.92
   885.5 1472.48   914.9 1483.83   924.8 1487.04   934.6 1488.45   954.2 1497.35
#Mann= 3 , 0 , 0
       0      .1       0   445.8    .045       0   460.8      .1       0
Bank Sta=445.8,460.8
XS Rating Curve= 0 ,0
Exp/Cntr=0.3,0.1

Type RM Length L Ch R = 1 ,49633.9 ,450.682,450.526,451.536
XS GIS Cut Line= 3
     1835348.747      347428.623     1835388.376      346982.805
     1835421.415      346366.488
#Sta/Elev= 30
       0 1538.62    38.9  1529.1    68.1 1519.36    77.8 1517.82    97.3 1509.86
     107 1508.52   136.2 1497.77   155.7 1493.05   175.1 1485.47   194.6 1481.12
   223.8 1470.24     253 1461.95   350.3  1442.5   379.5  1430.5   408.7 1413.53
   440.1  1408.5   455.1 1407.11   457.4 1407.05   486.8 1413.65   604.3 1415.24
   653.3 1424.77     859 1446.93   947.2 1461.73   966.8  1469.1   976.6 1470.42
   996.2 1478.08  1015.8 1482.63  1045.2 1494.81    1055 1495.96  1064.8 1499.66
#Mann= 3 , 0 , 0
       0      .1       0   440.1    .045       0   455.1      .1       0
Bank Sta=440.1,455.1
XS Rating Curve= 0 ,0
Exp/Cntr=0.3,0.1

Type RM Length L Ch R = 1 ,49183.4 ,373.725,377.873,379.088
XS GIS Cut Line= 3
     1835793.724      347406.272     1835796.766      346896.421
     1835827.266      346171.948
#Sta/Elev= 30
       0 1512.17    19.6 1506.44    39.2  1497.6    58.8 1492.83    78.4  1485.1
    98.1 1480.15   117.7 1473.15   137.3 1469.36   176.5 1458.71   196.1 1451.82
   215.7 1448.09   264.7 1434.81   343.2 1420.58   431.4  1407.6   460.8 1405.13
   503.5 1404.99   518.5 1404.94   539.3 1404.58   558.9 1406.21   588.3 1416.32
   627.4 1422.98     794 1439.05   862.6 1451.97   960.6 1465.79   980.2 1470.93
     990 1471.38  1058.6 1489.27  1068.4 1489.88    1137 1507.99    1235 1522.91
#Mann= 3 , 0 , 0
       0      .1       0   503.5    .045       0   518.5      .1       0
Bank Sta=503.5,518.5
XS Rating Curve= 0 ,0
Exp/Cntr=0.3,0.1

Type RM Length L Ch R = 1 ,48805.5 ,372.267,371.601,373.826
XS GIS Cut Line= 3
     1836061.389      347456.042     1836143.992      347022.375
     1836095.831      346492.856
#Sta/Elev= 30
       0 1515.07    19.6 1506.11    29.4 1503.83    49.1 1494.13    68.7 1488.15
    98.1 1476.33   107.9 1475.28   127.5 1468.22   147.2 1464.07   176.6 1453.55
   186.4 1452.81     206 1446.03   225.6 1442.06   255.1 1431.84   264.9 1430.54
   294.3  1420.9   372.8 1404.83   421.7 1402.11   436.7 1402.35   480.1 1407.21
   509.1 1408.51   625.1 1407.65   644.5  1413.1   654.1 1413.74   721.8 1432.56
   818.5 1450.05   847.5 1459.13   895.8  1470.3   924.8 1479.51   973.2 1489.08
#Mann= 3 , 0 , 0
       0      .1       0   421.7    .045       0   436.7      .1       0
Bank Sta=421.7,436.7
XS Rating Curve= 0 ,0
Exp/Cntr=0.3,0.1

Type RM Length L Ch R = 1 ,48433.9 ,399.695,400.408,399.47
XS GIS Cut Line= 3
     1836306.908      347446.522     1836438.562      346904.098
     1836558.469      346406.738
#Sta/Elev= 30
       0 1484.91    39.2 1472.59    58.8 1468.97    88.1 1459.34    97.9 1458.28
   137.1 1448.16   166.5  1438.8   244.8 1420.82   440.7 1404.56   499.4 1403.61
   548.4 1397.24   550.7 1397.29   565.7 1398.35   577.8 1401.67   607.4 1419.03
     627 1425.16   646.7 1435.07   666.4 1441.64   686.1 1451.29   774.6 1478.59
   823.8 1490.44   853.3 1501.74     873 1507.15   902.5 1517.72     932 1531.35
   981.2 1548.02  1020.6 1567.56  1030.4 1569.56  1050.1 1578.29  1069.8 1583.19
#Mann= 3 , 0 , 0
       0      .1       0   550.7    .045       0   565.7      .1       0
Bank Sta=550.7,565.7
XS Rating Curve= 0 ,0
Exp/Cntr=0.3,0.1

Type RM Length L Ch R = 1 ,48033.5 ,378.967,399.592,408.256
XS GIS Cut Line= 3
     1836655.886      347557.581     1836740.762      347110.792
      1836819.14      346661.322
#Sta/Elev= 30
       0 1490.98     9.7 1490.36    38.7 1477.36    77.4 1467.14    96.8 1463.62
   116.1 1457.38   174.2 1445.04   193.5 1438.89   222.6  1432.1   241.9 1425.49
   251.6 1424.47   270.9 1417.98     358 1404.26   406.4 1399.78   435.4 1393.08
   446.1  1393.3   461.1 1394.62   522.7 1400.53   610.1 1415.81   639.2 1424.44
   648.9 1425.01   716.9 1442.33   736.3 1445.33   765.4 1452.59   794.5 1462.22
     814 1465.83   852.8 1476.37   881.9 1486.17   891.6 1487.16     911 1495.12
#Mann= 3 , 0 , 0
       0      .1       0   446.1    .045       0   461.1      .1       0
Bank Sta=446.1,461.1
XS Rating Curve= 0 ,0
Exp/Cntr=0.3,0.1

Type RM Length L Ch R = 1 ,47633.9 ,395.888,400,410.144
XS GIS Cut Line= 3
     1836722.047      347600.929     1837123.576      347181.055
     1837339.984      346755.568
#Sta/Elev= 30
       0 1491.07    38.7 1481.57    58.1 1475.35    77.5 1472.73   116.2 1461.51
   164.6 1451.03   251.8 1437.58     426 1401.74   513.2 1395.55   542.2 1389.81
   561.6 1388.28   573.5 1389.23   588.5 1392.15   600.4 1394.47   658.9 1397.38
   707.6 1405.77   746.6 1414.93   775.8 1427.75   785.5 1429.27   814.8 1438.18
   834.3 1441.94     883 1459.13   902.5 1470.23   921.9 1477.25   951.2 1496.03
   970.6 1502.88   990.1 1512.46  1009.6 1517.97  1038.8 1535.89  1058.3  1542.8
#Mann= 3 , 0 , 0
       0      .1       0   573.5    .045       0   588.5      .1       0
Bank Sta=573.5,588.5
XS Rating Curve= 0 ,0
Exp/Cntr=0.3,0.1

Type RM Length L Ch R = 1 ,47233.9 ,491.342,506.371,530.026
XS GIS Cut Line= 3
     1836786.919      347681.118      1837393.18      347464.546
      1837737.45      347221.038
#Sta/Elev= 30
       0 1485.31    97.5 1466.06   146.3 1453.86   156.1 1452.68   175.6 1447.19
   185.3 1445.69   204.8 1439.82   214.6 1438.37   234.1 1433.15   282.9  1422.8
   302.4  1417.3   312.1 1416.24   331.6 1410.69   360.9 1405.88   429.2 1397.27
   507.2 1396.06     634 1382.83   636.3 1382.88   651.3 1384.52   692.8 1397.81
   761.5 1411.82   810.5 1415.63   839.9  1420.6   918.4  1427.1   947.8 1428.88
   967.4 1427.56   977.2 1429.63   996.8 1435.95  1016.4 1439.95  1065.5 1447.24
#Mann= 3 , 0 , 0
       0      .1       0   636.3    .045       0   651.3      .1       0
Bank Sta=636.3,651.3
XS Rating Curve= 0 ,0
Exp/Cntr=0.3,0.1

Type RM Length L Ch R = 1 ,46727.6 ,286.886,293.629,296.827
XS GIS Cut Line= 3
     1836784.836      347774.867     1837277.408      347911.175
     1837693.405      348084.661
#Sta/Elev= 30
       0 1483.43      59 1469.88   137.6 1448.73   186.7 1437.18   206.4 1430.96
   216.2 1429.25   235.9 1422.11   245.7  1420.5   294.9 1404.56   324.3 1398.44
   393.1 1386.07   507.6 1379.13   520.9  1378.4   522.6 1378.48   530.7 1378.91
   550.3 1384.59   569.9 1388.45   599.3 1397.44   618.9 1407.59   628.7 1410.35
   648.3 1421.42   658.1 1424.12   677.7 1434.01   716.8 1451.02     805  1474.3
   863.8 1498.09   883.4 1508.04   893.2 1509.73   942.2 1532.75   961.8 1540.41
#Mann= 3 , 0 , 0
       0      .1       0   507.6    .045       0   522.6      .1       0
Bank Sta=507.6,522.6
XS Rating Curve= 0 ,0
Exp/Cntr=0.3,0.1

Type RM Length L Ch R = 1 ,46433.9 ,407.227,400,393.382
XS GIS Cut Line= 3
     1836721.178      347892.345       1837106.7      348137.992
     1837502.901      348361.632
#Sta/Elev= 30
       0 1486.48    38.9 1476.91    97.3 1459.42     107 1457.87   165.3 1439.87
     214 1429.52   243.2 1422.02   252.9 1420.74   272.3 1414.71   282.1 1412.89
   311.2 1404.15   330.7 1399.64   379.3 1383.92   449.6 1373.83   464.6 1373.26
   466.8 1373.23   505.5 1376.79   573.3 1391.35   631.4 1411.37   641.1 1413.04
   660.4 1420.32   699.1 1432.64   708.8 1433.92   728.2 1440.83   747.5 1445.66
   766.9 1452.41   776.6 1454.08     854 1477.18   883.1  1490.3   912.1 1508.42
#Mann= 3 , 0 , 0
       0      .1       0   449.6    .045       0   464.6      .1       0
Bank Sta=449.6,464.6
XS Rating Curve= 0 ,0
Exp/Cntr=0.3,0.1

Type RM Length L Ch R = 1 ,46033.9 ,405.697,400,386.254
XS GIS Cut Line= 3
     1836473.779      348369.559     1836914.184      348480.819
     1837362.325      348581.439
#Sta/Elev= 30
       0 1480.09   154.6 1448.47   183.6 1443.83     232 1439.67   260.9 1434.63
   280.3  1426.3   289.9 1423.82   338.3 1402.08   347.9 1399.02   386.6 1380.69
   396.3 1374.98   405.9 1371.43   425.2 1367.31   434.9 1367.03   446.7 1368.93
   461.7 1374.57   483.6 1377.71   610.6 1374.29   659.5  1382.3   698.5 1393.71
   747.4 1411.88   757.2 1413.82   776.7 1421.61   786.5 1423.99     806  1432.4
   815.8 1433.84   835.4 1441.58   845.1 1443.32   864.7 1451.54   913.5 1466.98
#Mann= 3 , 0 , 0
       0      .1       0   446.7    .045       0   461.7      .1       0
Bank Sta=446.7,461.7
XS Rating Curve= 0 ,0
Exp/Cntr=0.3,0.1

Type RM Length L Ch R = 1 ,45633.9 ,395.233,400,407.844
XS GIS Cut Line= 3
      1836470.91      348873.236     1836949.985      348866.157
     1837368.373      348698.459
#Sta/Elev= 30
       0 1493.32     9.8 1491.67    29.3 1483.57    39.1 1481.93    58.7 1474.13
    68.4 1472.84      88 1464.92   117.3 1455.71   127.1  1454.4   146.7 1446.45
   195.6 1431.75   215.1 1423.24   224.9  1421.6   273.8  1407.3   283.6  1406.1
   332.5 1394.12   371.6 1387.21   420.5 1375.24   471.6 1368.55   486.6 1366.53
   518.3 1363.96   567.3 1369.52   577.1 1376.43   606.5 1385.16   655.5 1396.35
   684.9 1406.65   694.7 1408.07   802.5 1440.81   890.7 1460.68   929.9 1473.36
#Mann= 3 , 0 , 0
       0      .1       0   471.6    .045       0   486.6      .1       0
Bank Sta=471.6,486.6
XS Rating Curve= 0 ,0
Exp/Cntr=0.3,0.1

Type RM Length L Ch R = 1 ,45233.9 ,500.974,515.242,534.36
XS GIS Cut Line= 3
     1836428.391      349184.701     1836883.228      349214.024
      1837362.31      349163.947
#Sta/Elev= 30
       0 1479.76    58.2 1463.17   116.4 1445.06   135.8 1436.66   174.6 1425.71
   193.9  1418.9   300.6 1388.16     320 1381.47   329.7 1379.84   349.1 1373.32
   358.8 1371.89   378.2 1366.08     417 1361.36   448.3 1355.92   455.8 1355.71
   463.3 1355.99   524.6 1358.05   632.7 1378.88   652.4 1384.93   662.2 1386.34
   691.7 1394.12   711.4 1400.42   721.2  1401.9   740.9 1407.93   750.7 1409.53
   799.8 1425.06   809.7 1426.95   858.8 1442.84   898.2 1453.28   937.5 1461.62
#Mann= 3 , 0 , 0
       0      .1       0   448.3    .045       0   463.3      .1       0
Bank Sta=448.3,463.3
XS Rating Curve= 0 ,0
Exp/Cntr=0.3,0.1

Type RM Length L Ch R = 1 ,44718.7 ,287.644,284.758,277.042
XS GIS Cut Line= 3
     1836423.757      349371.074     1836796.815      349651.516
     1837133.317      349954.463
#Sta/Elev= 30
       0 1454.94    19.4 1448.04    68.1 1436.43   116.7 1421.61   155.6 1405.14
   204.2 1380.98   233.4 1370.02   252.8 1360.56     282 1350.61   379.2 1346.81
   447.8 1341.76     457 1341.32   462.8 1342.23   543.8 1354.31   582.3 1362.13
   601.6 1369.66   620.9 1374.85   649.8 1387.25   659.4 1388.55     669 1391.78
   726.8 1416.44   746.1 1422.53   765.4 1430.66   784.6 1434.05   823.2 1444.86
   842.4 1453.34   861.7 1459.54     881 1468.57   900.2 1473.11   919.5 1481.89
#Mann= 3 , 0 , 0
       0      .1       0   447.8    .045       0   462.8      .1       0
Bank Sta=447.8,462.8
XS Rating Curve= 0 ,0
Exp/Cntr=0.3,0.1

Type RM Length L Ch R = 1 ,44433.9 ,397.999,400,395.626
XS GIS Cut Line= 3
     1836198.213       349609.21      1836602.83      349839.583
     1837058.723       350053.02
#Sta/Elev= 30
       0 1491.21    48.5 1478.29    77.6 1468.19    87.3  1466.5   145.5 1448.87
   155.2 1447.41   223.1 1426.89   261.9 1413.22   358.9 1366.92   368.6 1364.38
   426.8 1341.19   458.1 1336.34   465.6 1336.19   473.1  1336.5   562.4  1343.3
   601.1  1341.9   639.9 1348.44   707.6 1371.57   746.3 1388.36   765.7 1398.33
   775.4 1400.64   794.7 1410.57   814.1 1417.61   833.5 1427.82   862.5 1439.13
   872.2 1440.37   881.9 1443.53   939.9 1462.78   959.3 1472.19     969 1474.42
#Mann= 3 , 0 , 0
       0      .1       0   458.1    .045       0   473.1      .1       0
Bank Sta=458.1,473.1
XS Rating Curve= 0 ,0
Exp/Cntr=0.3,0.1

Type RM Length L Ch R = 1 ,44033.9 ,411.504,400,398.62
XS GIS Cut Line= 3
     1836096.982      349970.939     1836530.147      350204.409
     1836966.481      350307.949
#Sta/Elev= 30
       0 1479.13     9.6 1473.48    28.9 1467.37    77.2 1444.42   115.8 1428.92
   183.3  1406.1   202.6 1402.54   221.9 1395.17   279.8 1378.53   299.1 1371.29
   318.4 1359.77   328.1 1356.25   405.2 1342.73   472.8 1332.05   482.4 1331.75
   484.6 1332.06   499.6 1336.06   521.3 1340.45   531.1 1345.06   540.8 1347.71
   560.3 1361.44   570.1 1364.54   589.6 1375.18   638.3 1388.51   696.8 1407.88
   716.3 1418.86   745.5 1429.71     882 1455.21     921 1472.78   940.5 1483.56
#Mann= 3 , 0 , 0
       0      .1       0   484.6    .045       0   499.6      .1       0
Bank Sta=484.6,499.6
XS Rating Curve= 0 ,0
Exp/Cntr=0.3,0.1

Type RM Length L Ch R = 1 ,43633.9 ,402.52,400,394.978
XS GIS Cut Line= 3
     1835915.967      350534.914     1836369.535      350529.099
     1836826.599      350602.367
#Sta/Elev= 30
       0 1453.42    19.3 1443.48    77.2  1423.5   183.4    1400   212.3 1391.96
   231.6 1385.14   241.3 1383.54   270.2 1375.38   289.5 1367.53   299.2 1366.22
   308.8 1362.05   318.5 1355.31   328.1 1353.02   337.8 1347.49   347.4 1344.47
   446.1 1327.59   461.1 1326.37   463.2 1326.33   530.8 1338.62   607.9 1348.16
   665.8 1358.46   685.1 1364.99   694.7 1366.44     714 1375.55   762.2 1391.69
   781.5 1400.88   820.1 1415.25   839.4 1424.34   868.3 1431.66   916.5 1440.66
#Mann= 3 , 0 , 0
       0      .1       0   446.1    .045       0   461.1      .1       0
Bank Sta=446.1,461.1
XS Rating Curve= 0 ,0
Exp/Cntr=0.3,0.1

Type RM Length L Ch R = 1 ,43233.9 ,456.968,472.63,487.517
XS GIS Cut Line= 3
     1835904.503       350984.84     1836355.802      350928.428
     1836810.994      350900.117
#Sta/Elev= 30
       0 1458.35      29  1450.6   106.4 1433.51   125.8 1427.71   135.5 1426.16
   154.8 1419.73   164.5 1418.31   183.9 1412.16   193.5 1411.07   212.9 1404.65
   222.6 1402.79   241.9 1393.63   251.6 1391.56     271 1380.47   280.6 1377.78
   309.7 1360.19   319.3 1353.16     329  1343.7   338.7 1338.88   348.4 1335.84
   425.8 1321.61   447.3 1319.43   462.3 1318.12   474.2 1317.67   571.3 1322.65
   590.7 1324.65   707.1 1344.65   804.1 1363.59   852.7 1376.74   910.9 1389.14
#Mann= 3 , 0 , 0
       0      .1       0   447.3    .045       0   462.3      .1       0
Bank Sta=447.3,462.3
XS Rating Curve= 0 ,0
Exp/Cntr=0.3,0.1

Type RM Length L Ch R = 1 ,42761.3 ,325.152,327.37,328.961
XS GIS Cut Line= 3
     1835948.831      351181.545     1836362.101      351389.381
     1836779.318      351643.078
#Sta/Elev= 30
       0 1414.67    19.3 1408.22    67.5 1397.09    86.7  1386.4   134.9 1370.28
   154.2  1360.9   163.8 1358.44   183.1 1348.53     212 1339.72   356.6 1313.34
     453 1309.94     474 1307.72     489 1306.16   491.9 1306.07   511.4 1307.23
   521.2 1309.56   530.9 1315.12   540.7 1317.69   550.5 1323.27     570 1338.29
   589.5 1349.21   599.3 1353.97   618.8 1359.74   667.7 1380.13     697    1389
   716.5 1396.41   794.6 1418.85   823.9  1428.5     863 1437.36   950.9 1460.89
#Mann= 3 , 0 , 0
       0      .1       0     474    .045       0     489      .1       0
Bank Sta=474,489
XS Rating Curve= 0 ,0
Exp/Cntr=0.3,0.1

Type RM Length L Ch R = 1 ,42433.9 ,402.101,401.028,398.317
XS GIS Cut Line= 3
     1835834.177      351390.901     1836196.431      351666.214
     1836558.685      351941.527
#Sta/Elev= 30
       0 1392.38    58.1 1375.28    67.8 1374.22   106.5 1363.63   125.9 1356.11
   145.2 1351.75   164.6 1343.25   203.3 1330.45   309.8 1311.42   387.2 1304.31
   447.5 1301.48     455 1300.65   462.5  1300.8   493.7 1303.21   522.8 1310.61
   532.4 1315.86   551.8 1330.85   561.5 1334.57   590.5 1350.06   600.2 1353.22
   629.3 1369.41     697 1394.58   716.4 1400.55   774.5 1425.94   793.8 1432.37
   813.2 1441.13   832.6 1447.28   861.6  1460.7   871.3 1463.34     910 1487.01
#Mann= 3 , 0 , 0
       0      .1       0   447.5    .045       0   462.5      .1       0
Bank Sta=447.5,462.5
XS Rating Curve= 0 ,0
Exp/Cntr=0.3,0.1

Type RM Length L Ch R = 1 ,42032.9 ,433.776,438.109,444.368
XS GIS Cut Line= 3
     1835552.653      351696.534     1835925.065      351957.295
      1836320.95      352185.827
#Sta/Elev= 30
       0 1438.22    87.1 1410.13   116.1 1399.66   135.4  1390.8   154.8 1385.41
   212.8 1361.05   222.5 1358.04   251.5 1342.57   280.5 1329.11   328.9 1314.57
   396.6 1298.42   415.9 1294.01   435.3 1292.61     441 1293.04     456 1295.46
   571.3  1313.2   590.8 1315.14     620 1321.22   658.9 1325.98     688 1331.75
   697.8 1334.53   717.2 1344.22   765.9 1363.43   785.3 1374.75   804.8 1381.44
   824.2  1391.2   833.9 1393.57   853.4 1403.85   892.3 1415.64   911.7 1418.76
#Mann= 3 , 0 , 0
       0      .1       0     441    .045       0     456      .1       0
Bank Sta=441,456
XS Rating Curve= 0 ,0
Exp/Cntr=0.3,0.1

Type RM Length L Ch R = 1 ,41594.8 ,347.425,360.863,371.108
XS GIS Cut Line= 3
     1835343.635      351978.982     1835665.299      352307.648
     1835970.262      352644.159
#Sta/Elev= 30
       0 1404.57     9.8 1402.97    48.9 1388.14    68.5 1382.91   107.6 1369.15
   117.4 1367.45     137 1359.57   156.6  1349.8   176.1 1344.96   205.5 1331.53
   244.6 1319.69   322.9 1301.29   352.2 1296.14   437.4 1287.09   452.4 1285.42
   459.9 1284.91   469.5 1285.66   479.2 1288.09   537.2 1304.67   556.5 1311.34
   595.2 1330.54   614.5 1335.06   633.8 1343.45   662.8 1350.46   701.4  1364.1
   749.8 1372.64   807.7  1375.9   827.1 1373.82   875.4 1374.05     914 1377.34
#Mann= 3 , 0 , 0
       0      .1       0   437.4    .045       0   452.4      .1       0
Bank Sta=437.4,452.4
XS Rating Curve= 0 ,0
Exp/Cntr=0.3,0.1

Type RM Length L Ch R = 1 ,41233.9 ,406.193,400,396.712
XS GIS Cut Line= 3
     1835263.712      351994.315      1835354.14      352445.218
     1835500.306      352891.112
#Sta/Elev= 30
       0 1413.07    19.6 1404.84    39.1 1399.68    58.7 1391.84    78.3 1387.04
    97.8 1378.72   117.4 1373.34     137 1365.63   195.7 1353.47   234.8 1339.16
   254.4 1325.53   264.2 1321.89   313.1 1312.06   342.5 1303.72   381.6 1295.28
   430.5 1286.36   452.4 1279.72   459.9  1278.7   467.4 1278.98   528.3  1289.1
   557.6 1296.25     587 1306.97   596.7  1308.2   616.3 1314.42   694.5 1332.99
   723.8 1336.74   782.5 1348.18   850.9 1358.75   880.2 1365.37   929.1 1370.57
#Mann= 3 , 0 , 0
       0      .1       0   452.4    .045       0   467.4      .1       0
Bank Sta=452.4,467.4
XS Rating Curve= 0 ,0
Exp/Cntr=0.3,0.1

Type RM Length L Ch R = 1 ,40833.9 ,326.436,326.104,325.772
XS GIS Cut Line= 3
     1834773.706      352166.748     1834981.227      352571.668
     1835188.749      352976.587
#Sta/Elev= 30
       0 1422.94      29  1416.6    67.8 1404.51    96.8  1391.9   116.2 1387.07
   135.5 1377.94   154.9 1372.04   183.9 1358.29   203.3 1352.49   222.7 1343.96
     242 1338.93   271.1 1322.03   309.8 1312.49   329.1 1309.38   358.2  1299.7
   416.3 1285.24   435.6 1275.64   447.5  1272.8     455 1272.45   462.5 1272.91
   590.5  1288.3   648.6 1297.64   716.4 1317.83   735.7 1322.12   755.1  1328.9
   813.2 1344.22   842.2 1355.19   861.6 1359.23     881 1366.12     910 1373.27
#Mann= 3 , 0 , 0
       0      .1       0   447.5    .045       0   462.5      .1       0
Bank Sta=447.5,462.5
XS Rating Curve= 0 ,0
Exp/Cntr=0.3,0.1

Type RM Length L Ch R = 1 ,40507.8 ,374.977,377.299,379.62
XS GIS Cut Line= 3
     1834475.744      352290.422     1834679.028      352697.684
     1834892.478      353099.474
#Sta/Elev= 30
       0 1392.27    19.4 1389.33    48.4 1381.07    67.8 1377.52    87.2 1370.56
   106.5 1366.04   135.6 1353.92   193.7 1342.51   232.4 1325.99   242.1 1324.15
   261.5    1317   280.9  1313.2   309.9  1303.9   329.3 1300.26   348.6 1294.11
   416.4 1285.78   470.6 1271.42   474.5 1270.56   485.6 1270.93   513.3 1272.26
   542.3 1276.48   571.3 1285.87   629.4 1291.28   677.8 1298.61   706.9 1304.91
   726.2 1306.35   745.6 1315.94   832.7 1345.37   900.5 1361.51   910.1 1364.89
#Mann= 3 , 0 , 0
       0      .1       0   470.6    .045       0   485.6      .1       0
Bank Sta=470.6,485.6
XS Rating Curve= 0 ,0
Exp/Cntr=0.3,0.1

Type RM Length L Ch R = 1 ,40130.5 ,613.407,590.829,566.955
XS GIS Cut Line= 3
     1834252.741      352373.066     1834324.972      352815.301
     1834510.772      353273.166
#Sta/Elev= 30
       0 1345.12    87.7 1339.12   126.6 1332.76   136.4  1332.2   155.9  1326.6
   175.3 1323.21   204.6 1313.75   214.3 1312.51   233.8 1305.61   253.3 1301.25
   282.5 1291.91   311.7 1286.69   379.9 1278.07   469.8 1264.08   484.8 1262.91
   486.9 1262.88   496.5 1263.89   515.9 1268.46   583.7 1275.14   661.2 1286.98
   670.9  1289.4   690.3 1296.13     700 1297.72   729.1 1309.82   738.8 1311.76
   767.8 1320.75   816.3 1328.47   874.4 1331.33   922.8 1332.01   942.2 1333.25
#Mann= 3 , 0 , 0
       0      .1       0   469.8    .045       0   484.8      .1       0
Bank Sta=469.8,484.8
XS Rating Curve= 0 ,0
Exp/Cntr=0.3,0.1

Type RM Length L Ch R = 1 ,39539.7 ,312.818,305.768,300.534
XS GIS Cut Line= 3
     1833587.886      353117.846     1834038.212      353239.831
     1834479.201      353345.371
#Sta/Elev= 30
       0 1363.14    19.4 1355.51    29.2 1354.27    48.6  1347.1   116.6 1329.54
   165.2 1318.74   184.7 1312.44   194.4 1310.72   223.6 1302.26     243 1294.24
   272.2 1286.86   349.9 1275.11   408.2 1264.33   427.7  1258.4   437.4 1256.83
   449.7 1257.51   464.7  1259.1   505.1  1261.5   611.3 1262.38   630.6  1265.9
   649.9 1272.85   659.5 1274.01   678.8 1279.87   784.9 1298.02   804.2  1302.8
   813.9 1304.11   833.2 1309.98   871.8 1317.66   900.7 1325.52     920 1328.75
#Mann= 3 , 0 , 0
       0      .1       0   449.7    .045       0   464.7      .1       0
Bank Sta=449.7,464.7
XS Rating Curve= 0 ,0
Exp/Cntr=0.3,0.1

Type RM Length L Ch R = 1 ,39233.9 ,401.901,400,389.963
XS GIS Cut Line= 3
     1833479.069      353526.098     1833923.733      353511.275
     1834435.685      353526.368
#Sta/Elev= 30
       0 1419.02     9.7 1415.12    19.3 1413.64    38.7 1405.63    48.4 1403.83
    67.7 1395.47    77.4 1393.65    96.7 1383.95   125.7 1373.18   135.4 1370.97
   164.4 1358.63   222.5 1338.18   261.1 1327.22   280.5 1318.97   299.8 1312.51
   338.5 1295.62   357.9 1289.13   377.2 1280.15   386.9 1277.14   437.4 1250.46
   452.4 1248.49   454.6  1248.3   531.9 1257.19   686.5 1258.52   754.1 1260.34
   773.5  1263.5   841.1 1280.51   899.1 1298.07   918.4 1306.13   957.1 1318.85
#Mann= 3 , 0 , 0
       0      .1       0   437.4    .045       0   452.4      .1       0
Bank Sta=437.4,452.4
XS Rating Curve= 0 ,0
Exp/Cntr=0.3,0.1

Type RM Length L Ch R = 1 ,38833.9 ,330.871,341.861,359.029
XS GIS Cut Line= 3
     1833580.521      353932.484     1834079.443      353871.254
     1834488.589      353692.253
#Sta/Elev= 30
       0 1348.28    38.7 1340.36    67.7  1332.8   164.3 1314.74   183.7 1309.29
   193.3  1307.9   212.7 1300.38     232 1295.46   280.3 1288.43   338.3 1271.34
   367.3  1266.1   444.7 1260.48   473.7 1252.67   495.2 1244.91   510.2 1242.01
   522.1 1241.02   531.8 1241.69   560.9 1247.34   696.8 1259.12   716.3 1265.03
   764.8 1275.57   784.2 1284.02   803.6 1290.16   813.3 1294.92   832.8 1300.26
   852.2 1307.31   900.7 1319.31   920.1 1325.65   929.8 1326.64   949.3 1331.05
#Mann= 3 , 0 , 0
       0      .1       0   495.2    .045       0   510.2      .1       0
Bank Sta=495.2,510.2
XS Rating Curve= 0 ,0
Exp/Cntr=0.3,0.1

Type RM Length L Ch R = 1 ,38492.1 ,457.188,458.44,459.552
XS GIS Cut Line= 3
     1833584.267      353982.733       1834045.7       354173.56
     1834506.575      354322.271
#Sta/Elev= 30
       0 1332.97    39.2 1326.26    68.5 1317.16   146.9 1297.54   195.8 1282.41
     235 1274.25   264.4 1265.59   303.5 1257.58   332.9 1249.93   352.5 1248.26
   401.4 1249.21   450.4  1248.7     470 1247.31     509 1241.17     524 1238.15
   538.1 1237.08   547.8 1238.99   557.4 1242.81   567.1 1245.29   586.5 1253.49
   615.6 1262.54   634.9  1266.8   673.7 1277.56   712.4 1290.35   722.1 1292.29
   751.2 1300.86   809.3 1310.76   886.8 1318.71   935.2 1326.96   983.6 1332.89
#Mann= 3 , 0 , 0
       0      .1       0     509    .045       0     524      .1       0
Bank Sta=509,524
XS Rating Curve= 0 ,0
Exp/Cntr=0.3,0.1

Type RM Length L Ch R = 1 ,38033.6 ,395.69,400.336,403.829
XS GIS Cut Line= 3
     1833335.854      354346.664     1833757.027      354518.704
     1834183.495      354678.017
#Sta/Elev= 30
       0 1361.73    19.4 1356.76    38.7 1348.45    48.4 1346.09    67.8 1336.08
    96.8 1326.52   116.2 1322.06   154.9 1309.87   164.6 1306.02   174.2 1304.01
   203.3 1293.95   251.7 1279.93     271 1272.84   280.7 1270.83   300.1 1257.82
   329.1 1240.07   338.8 1237.99   406.6 1236.55   416.2  1235.5   435.6 1231.35
   445.3 1230.95   445.4 1230.95   460.4 1231.73     484 1232.84   503.4 1235.03
   532.4 1240.67   590.6 1247.83   755.2 1257.42   832.7 1260.41   910.2 1271.63
#Mann= 3 , 0 , 0
       0      .1       0   445.4    .045       0   460.4      .1       0
Bank Sta=445.4,460.4
XS Rating Curve= 0 ,0
Exp/Cntr=0.3,0.1

Type RM Length L Ch R = 1 ,37633.3 ,399.366,412.884,427.77
XS GIS Cut Line= 3
     1833215.603      354621.189     1833593.242      354879.569
     1833991.321      355098.989
#Sta/Elev= 30
       0  1320.3    19.5 1315.44    48.7 1306.16    68.1 1302.29    87.6 1296.84
    97.4 1293.82   116.8 1286.06   136.3 1281.46   175.2 1268.86     185 1266.72
   214.2 1262.41   262.9 1252.04   292.1 1247.69   301.8 1246.62   360.2 1244.38
   418.6 1240.17   428.4 1238.24   438.1 1234.15   447.8 1228.79     455 1226.37
     470 1223.83   476.9  1223.5   496.3 1223.86   534.9 1227.42   631.7 1231.93
     651 1233.56     680 1236.58     709 1242.01   728.4 1246.83   912.1 1265.61
#Mann= 3 , 0 , 0
       0      .1       0     455    .045       0     470      .1       0
Bank Sta=455,470
XS Rating Curve= 0 ,0
Exp/Cntr=0.3,0.1

Type RM Length L Ch R = 1 ,37220.4 ,348.142,355.225,362.308
XS GIS Cut Line= 3
     1833156.127       354733.39     1833257.606      354920.735
     1833606.277       355610.27
#Sta/Elev= 30
       0 1294.47     9.7  1293.1    38.7  1283.1    77.5 1272.61   310.9 1228.43
   408.7  1224.4   477.1 1228.68   486.9 1228.32   517.2 1221.74   532.2 1216.59
   545.6 1211.77   555.4 1211.55     575  1217.5   584.7 1227.02   604.3 1240.67
   633.6 1251.49   653.2    1261     663 1262.71   692.3 1275.03   711.9 1280.15
   741.2 1291.13     751 1292.21   829.2 1318.15     839 1319.01   868.4 1329.91
   897.7 1337.15   917.3 1344.54   927.1 1345.65   956.4  1356.5   985.7 1363.64
#Mann= 3 , 0 , 0
       0      .1       0   517.2    .045       0   532.2      .1       0
Bank Sta=517.2,532.2
XS Rating Curve= 0 ,0
Exp/Cntr=0.3,0.1

Type RM Length L Ch R = 1 ,36865.2 ,311.513,307.281,303.049
XS GIS Cut Line= 3
     1832982.574      354819.863     1833066.007      355267.148
     1833149.439      355714.433
#Sta/Elev= 30
       0 1284.93      29 1277.78    87.1 1268.45   116.2 1261.47   125.9 1258.23
   145.2 1248.18   164.6 1241.83   183.9 1232.01   193.6 1229.29   222.7 1226.34
   319.5  1225.2   377.6 1220.29   445.3 1219.48     455 1218.61   480.4 1208.41
   493.7 1205.86   495.4  1206.3   522.8 1212.75   561.5 1216.56   571.2 1219.73
   580.9 1225.41   590.5 1227.67   629.3  1243.8   716.4 1262.32   755.1 1272.91
   784.1 1282.78   832.6 1291.66   861.6 1299.74   900.3  1307.7     910 1308.47
#Mann= 3 , 0 , 0
       0      .1       0   480.4    .045       0   495.4      .1       0
Bank Sta=480.4,495.4
XS Rating Curve= 0 ,0
Exp/Cntr=0.3,0.1

Type RM Length L Ch R = 1 ,36557.9 ,643.165,631.87,620.456
XS GIS Cut Line= 3
      1832619.65      354932.175     1832768.279      355362.135
     1832933.948      355786.365
#Sta/Elev= 30
       0 1304.87    48.4 1297.76    77.4 1291.38   135.5 1282.53   174.2 1274.69
   183.9 1271.73   203.3 1262.22   212.9 1261.03     242 1250.88     271 1242.95
   300.1 1239.53   348.5 1217.48   358.1 1214.25   367.8  1212.8   435.6 1211.11
   454.9 1201.16   470.6 1200.26   474.3 1200.17   485.6 1203.92   503.4 1207.78
   532.4 1210.21   668.1 1215.81   677.8 1217.76   706.9 1228.81   726.2 1230.85
   745.6 1237.05   755.3 1241.09   774.7 1252.42   784.4 1256.15   910.4    1280
#Mann= 3 , 0 , 0
       0      .1       0   470.6    .045       0   485.6      .1       0
Bank Sta=470.6,485.6
XS Rating Curve= 0 ,0
Exp/Cntr=0.3,0.1
